--- K120-00-00.prj (project) ---

Proj Title=K120-00-00
Current Plan=p02
Default Exp/Contr=.3,.1
English Units
Geom File=g01
Flow File=f02
Flow File=f01
Flow File=f04
Plan File=p02
Plan File=p01
Plan File=p04
Y Axis Title=Elevation
X Axis Title(PF)=Main Channel Distance
X Axis Title(XS)=Station
BEGIN DESCRIPTION:
Cypress Creek Watershed
Lemm Gully
HCFCD Unit K120-00-00
Flood Hazard Model
10, 2, 1, 0.2%
Filename k120-00-00
Prepared by:  Halff Associates  DATE:  03-26-04
Reviewed by:  _________  DATE:  __________________
STATUS (Final)
END DESCRIPTION:
DSS Export Rating Curves= 0
DSS Export Rating Curve Sorted= 0
DSS Export Volume Flow Curves= 0
DXF OffsetX= 0
DXF OffsetY= 0
DXF ScaleX= 1
DXF ScaleY= 10

--- K120-00-00.p02 (plan) ---

Plan Title=Floodway
Version=Version 3.0.1  Mar 2001
Short Identifier=Floodway0607
Geom File=g01
Flow File=f02
Subcritical Flow
K Sum by GR= 0
Std Step Tol= 0.01
Critical Tol= 0.01
Num of Std Step Trials= 20
Max Error Tol= 0.3
Flow Tol Ratio= 0.001
Split Flow NTrial= 30
Split Flow Tol= 0.02
Split Flow Ratio= 0.02
Log Output Level= 0
Friction Slope Method= 1
Unsteady Friction Slope Method= 2
Parabolic Critical Depth
Global Vel Dist= 0 , 0 , 0
Global Log Level= 0
CheckData=True
Encroach Param=-1 ,0,0, 3
Encroach River=K120-00-00
Encroach Reach=Reach - 1
Encroach Node=16297.90
       1  4978.4  5025.7       4       1
Encroach Node=15732.
       1  4965.4  5035.4       0       0       0
Encroach Node=15632.90
       1  4990.5  5011.7       4       1
Encroach Node=15612.80
       1  4990.5  5011.7       4       1
Encroach Node=15592.70
       1  4990.5  5011.7       4       1
Encroach Node=15484.
       1  4959.9  5059.9       0       0       0
Encroach Node=15361.
       1  4958.3  5048.3       0       0       0
Encroach Node=15263.90
       1  4944.9  5034.4       4       1
Encroach Node=15213.75
       1  4944.9  5034.4       4       1
Encroach Node=15163.60
       1  4944.9  5034.4       4       1
Encroach Node=15060.
       1  4967.3  5049.9       0       0       0
Encroach Node=13676.60
       1  4968.7  5040.6       4       1
Encroach Node=13330.
       1  4942.7  5042.2       0       0       0
Encroach Node=13233.60
       1  4960.9  5042.7       4       1
Encroach Node=13223.60
       1  4960.9  5042.7       4       1
Encroach Node=13213.60
       1  4959.9  5042.8       4       1
Encroach Node=13185.50
       1  4973.9  5065.2       4       1
Encroach Node=13058.10
       1  4973.9  5065.2       4       1
Encroach Node=12930.70
       1  4973.9  5065.2       4       1
Encroach Node=12832.
       1  4937.9  5048.2       0       0       0
Encroach Node=11782.60
       1  4960.2  5039.8       4       1
Encroach Node=11669.
       1  4942.2  5052.2       0       0       0
Encroach Node=11558.80
       1  4958.1  5037.7       4       1
Encroach Node=11547.80
       1  4961.3  5067.4       4       1
Encroach Node=11536.80
       1  4961.3  5067.4       4       1
Encroach Node=11427.
       1  4910.7  5061.8       0       0       0
Encroach Node=11164.70
       1  4937.9 5360.61       4       1
Encroach Node=10777.
       1  4930.3  5078.8       0       0       0
Encroach Node=10686.10
       1  4984.7  5014.7       4       1
Encroach Node=10659.50
       1  4984.7  5014.7       4       1
Encroach Node=10632.90
       1  4984.7  5014.7       4       1
Encroach Node=10520.
       1    4939  5079.3       0       0       0
Encroach Node=9867.
       1  4930.1    5068       0       0       0
Encroach Node=9710.30
       1 2659.91  2796.4       4       1
Encroach Node=9611.90
       1 2659.91  2796.4       4       1
Encroach Node=9513.50
       1 2659.91  2796.4       4       1
Encroach Node=9303.
       1    4932    5062       0       0       0
Encroach Node=7601.60
       1    4966  5038.2       4       1
Encroach Node=5849.00
       1  4961.8  5044.3       4       1
Encroach Node=4542.
       1  4940.5  5080.5       0       0       0
Encroach Node=4441.90
       1  4953.4  5050.6       4       1
Encroach Node=4418.30
       1  4953.4  5050.6       4       1
Encroach Node=4394.70
       1  4953.4  5050.6       4       1
Encroach Node=4294.
       1  4931.5  5071.5       0       0       0
Encroach Node=3707.20
       1  4945.4  5049.3       4       1
Encroach Node=2576.00
       1  4940.7  5035.3       4       1
Encroach Node=2462.
       1    4935  5059.5       0       0       0
Encroach Node=2362.40
       1    4963  5048.8       4       1
Encroach Node=2350.85
       1    4963  5048.8       4       1
Encroach Node=2339.30
       1    4963  5048.8       4       1
Encroach Node=2243
       1  4951.9  5051.9       0       0       0
Encroach Reach=K120-00-00_0022
Encroach Node=16297.90
       1  4978.4  5025.7       0       0       0
Encroach Node=15732.
       1  4965.4  5035.4       0       0       0
Encroach Node=15632.90
       1  4990.5  5011.7       0       0       0
Encroach Node=15612.80
       1  4990.5  5011.7       0       0       0
Encroach Node=15592.70
       1  4990.5  5011.7       0       0       0
Encroach Node=15484.
       1  4959.9  5059.9       0       0       0
Encroach Node=15361.
       1  4958.3  5048.3       0       0       0
Encroach Node=15263.90
       1  4944.9  5034.4       0       0       0
Encroach Node=15213.75
       1  4944.9  5034.4       0       0       0
Encroach Node=15163.60
       1  4944.9  5034.4       0       0       0
Encroach Node=15060.
       1  4967.3  5049.9       0       0       0
Encroach Node=13676.60
       1  4968.7  5040.6       0       0       0
Encroach Node=13330.
       1  4942.7  5042.2       0       0       0
Encroach Node=13233.60
       1  4960.9  5042.7       0       0       0
Encroach Node=13223.60
       1  4960.9  5042.7       0       0       0
Encroach Node=13213.60
       1  4959.9  5042.8       0       0       0
Encroach Node=13185.50
       1  4973.9  5065.2       0       0       0
Encroach Node=13058.10
       1  4973.9  5065.2       0       0       0
Encroach Node=12930.70
       1  4973.9  5065.2       0       0       0
Encroach Node=12832.
       1  4937.9  5048.2       0       0       0
Encroach Node=11782.60
       1  4960.2  5039.8       0       0       0
Encroach Node=11669.
       1  4942.2  5052.2       0       0       0
Encroach Node=11558.80
       1  4958.1  5037.7       0       0       0
Encroach Node=11547.80
       1  4961.3  5067.4       0       0       0
Encroach Node=11536.80
       1  4961.3  5067.4       0       0       0
Encroach Node=11427.
       1  4910.7  5061.8       0       0       0
Encroach Node=11164.70
       1  4937.9 5360.61       0       0       0
Encroach Node=10777.
       1  4930.3  5078.8       0       0       0
Encroach Node=10686.10
       1  4984.7  5014.7       0       0       0
Encroach Node=10659.50
       1  4984.7  5014.7       0       0       0
Encroach Node=10632.90
       1  4984.7  5014.7       0       0       0
Encroach Node=10520.
       1    4939  5079.3       0       0       0
Encroach Node=9867.
       1  4930.1    5068       0       0       0
Encroach Node=9710.30
       1 2659.91  2796.4       0       0       0
Encroach Node=9611.90
       1 2659.91  2796.4       0       0       0
Encroach Node=9513.50
       1 2659.91  2796.4       0       0       0
Encroach Node=9303.
       1    4932    5062       0       0       0
Encroach Node=7601.60
       1    4966  5038.2       0       0       0
Encroach Node=5849.00
       1  4961.8  5044.3       0       0       0
Encroach Node=4542.
       1  4940.5  5080.5       0       0       0
Encroach Node=4441.90
       1  4953.4  5050.6       0       0       0
Encroach Node=4418.30
       1  4953.4  5050.6       0       0       0
Encroach Node=4394.70
       1  4953.4  5050.6       0       0       0
Encroach Node=4294.
       1  4931.5  5071.5       0       0       0
Encroach Node=3707.20
       1  4945.4  5049.3       0       0       0
Encroach Node=2576.00
       1  4940.7  5035.3       0       0       0
Encroach Node=2462.
       1    4935  5059.5       0       0       0
Encroach Node=2362.40
       1    4963  5048.8       0       0       0
Encroach Node=2350.85
       1    4963  5048.8       0       0       0
Encroach Node=2339.30
       1    4963  5048.8       0       0       0
Encroach Node=2243
       1  4951.9  5051.9       0       0       0
Computation Interval=1HOUR
Output Interval=1HOUR
Run HTab= 0
Run UNet= 0
Run PostProcess= 0
UNET Theta= 1
UNET ZTol= 0.02
UNET ZSATol= 0.1
UNET MxIter= 20
UNET MaxInSteps= 20
UNET DtIC= 0
UNET DtMin= 0
UNET MaxCRTS= 20
UNET WFStab= 2
UNET SFStab= 1
UNET WFX= 1
UNET SFX= 1
UNET Convert EG Bridges=-1
UNET Use Existing IB Tables=-1
Instantaneous Interval=1HOUR
Write IC File= 0
Write Velocity= 0
Write Detailed= 0

--- K120-00-00.p01 (plan) ---

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Plan Title=FEMA Effective June 2007
Short Identifier=FEMAeff0607
Geom File=g01
Flow File=f01
Persistent XS Scale= 4902.95358649789 , 5084.38818565401 , 119.924050632911 , 102.759493670886 , 50 , 2
Encroach Param=-1 ,0,0, 0
IC Time=0

--- K120-00-00.p04 (plan) ---

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Plan Title=Storage Routing
Short Identifier=Store_Rout
Geom File=g01
Flow File=f04
Encroach Param=-1 ,0,0, 0

--- K120-00-00.f02 (steady flow) ---

Flow Title=Floodway
Version=Version 3.0.1  Mar 2001
Number of Profiles= 2
Profile Names=1PCT_100yr, 1PCTFloodway_100yrFW
River Rch & RM=K120-00-00,K120-00-00_0022,16297.90
     510     510
River Rch & RM=K120-00-00,K120-00-00_0022,15592.70
     530     530
River Rch & RM=K120-00-00,K120-00-00_0022,15163.60
     610     610
River Rch & RM=K120-00-00,K120-00-00_0022,13676.6
     660     660
River Rch & RM=K120-00-00,K120-00-00_0022,12930.70
     760     760
River Rch & RM=K120-00-00,K120-00-00_0022,11164.7
    1790    1790
River Rch & RM=K120-00-00,K120-00-00_0022,9513.50
    1900    1900
River Rch & RM=K120-00-00,K120-00-00_0022,7601.6
    2000    2000
River Rch & RM=K120-00-00,K120-00-00_0022,5849
    2060    2060
River Rch & RM=K120-00-00,K120-00-00_0022,4394.70
    2090    2090
River Rch & RM=K120-00-00,K120-00-00_0022,3707.2
    2140    2140
River Rch & RM=K120-00-00,K120-00-00_0022,2576.0
    2150    2150
River Rch & RM=K120-00-00,K120-00-00_0022,2339.30
    2254    2254
Boundary for River Rch & Prof#=K120-00-00,K120-00-00_0022, 1
Up Type= 0
Dn Type= 3
Dn Slope=.005
Boundary for River Rch & Prof#=K120-00-00,K120-00-00_0022, 2
Up Type= 0
Dn Type= 1
Dn Known WS=81.77
DSS Import GetInterval= 0
DSS Import GetPeak= 0
DSS Import FillOption= 0

--- K120-00-00.f01 (steady flow) ---

Flow Title=FEMA Effective June 2007
Version=Version 3.0.1  Mar 2001
Number of Profiles= 4
Profile Names=10PCT_10yr, 2PCT_50yr, 1PCT_100yr, 0.2PCT_500yr
River Rch & RM=K120-00-00,K120-00-00_0022,16297.90
     270     410     510     740
River Rch & RM=K120-00-00,K120-00-00_0022,15592.70
     280     430     530     770
River Rch & RM=K120-00-00,K120-00-00_0022,15163.60
     320     510     610     910
River Rch & RM=K120-00-00,K120-00-00_0022,13676.60
     350     550     660     990
River Rch & RM=K120-00-00,K120-00-00_0022,12930.70
     400     640     760    1150
River Rch & RM=K120-00-00,K120-00-00_0022,11164.70
     930    1560    1790    2550
River Rch & RM=K120-00-00,K120-00-00_0022,9513.50
     990    1630    1900    2720
River Rch & RM=K120-00-00,K120-00-00_0022,7601.60
    1050    1700    2000    2900
River Rch & RM=K120-00-00,K120-00-00_0022,5849.00
    1090    1750    2060    3000
River Rch & RM=K120-00-00,K120-00-00_0022,4394.70
    1100    1770    2090    3040
River Rch & RM=K120-00-00,K120-00-00_0022,3707.20
    1130    1810    2140    3120
River Rch & RM=K120-00-00,K120-00-00_0022,2576.00
    1140    1810    2150    3140
River Rch & RM=K120-00-00,K120-00-00_0022,2339.30
    1205    1895    2254    3311
Boundary for River Rch & Prof#=K120-00-00,K120-00-00_0022, 1
Up Type= 0
Dn Type= 3
Dn Slope=.005
Boundary for River Rch & Prof#=K120-00-00,K120-00-00_0022, 2
Up Type= 0
Dn Type= 3
Dn Slope=.005
Boundary for River Rch & Prof#=K120-00-00,K120-00-00_0022, 3
Up Type= 0
Dn Type= 3
Dn Slope=.005
Boundary for River Rch & Prof#=K120-00-00,K120-00-00_0022, 4
Up Type= 0
Dn Type= 3
Dn Slope=.005
DSS Import GetInterval= 0
DSS Import GetPeak= 0
DSS Import FillOption= 0

--- K120-00-00.f04 (steady flow) ---

Flow Title=Storage Routing
Version=Version 3.0.1  Mar 2001
Number of Profiles= 7
Profile Names=0.25*10% flood, 0.50*10%flood, 10% flood, 2% flood, 1% flood, 0.2%flood, 1.25*0.2% flood
River Rch & RM=K120-00-00,K120-00-00_0022,16297.90
      79     159     317     719     941    1541    1926
River Rch & RM=K120-00-00,K120-00-00_0022,15263.90
     113     226     451    1052    1383    2307    2884
River Rch & RM=K120-00-00,K120-00-00_0022,11782.6
     135     269     538    1270    1672    2808    3510
River Rch & RM=K120-00-00,K120-00-00_0022,11164.7
     299     598    1195    2667    3399    5533    6916
River Rch & RM=K120-00-00,K120-00-00_0022,10686.10
     315     631    1261    2779    3533    5760    7200
River Rch & RM=K120-00-00,K120-00-00_0022,9710.30
     338     675    1350    2929    3715    6066    7583
River Rch & RM=K120-00-00,K120-00-00_0022,5849
     367     734    1467    3129    3950    6471    8089
River Rch & RM=K120-00-00,K120-00-00_0022,4441.90
     369     738    1475    3143    3967    6499    8124
River Rch & RM=K120-00-00,K120-00-00_0022,3707.2
     382     764    1528    3234    4076    6684    8355
Boundary for River Rch & Prof#=K120-00-00,K120-00-00_0022, 1
Up Type= 0
Dn Type= 3
Dn Slope=.005
Boundary for River Rch & Prof#=K120-00-00,K120-00-00_0022, 2
Up Type= 0
Dn Type= 3
Dn Slope=.005
Boundary for River Rch & Prof#=K120-00-00,K120-00-00_0022, 3
Up Type= 0
Dn Type= 3
Dn Slope=.005
Boundary for River Rch & Prof#=K120-00-00,K120-00-00_0022, 4
Up Type= 0
Dn Type= 3
Dn Slope=.005
Boundary for River Rch & Prof#=K120-00-00,K120-00-00_0022, 5
Up Type= 0
Dn Type= 3
Dn Slope=.005
Boundary for River Rch & Prof#=K120-00-00,K120-00-00_0022, 6
Up Type= 0
Dn Type= 3
Dn Slope=.005
Boundary for River Rch & Prof#=K120-00-00,K120-00-00_0022, 7
Up Type= 0
Dn Type= 3
Dn Slope=.005
DSS Import GetInterval= 0
DSS Import GetPeak= 0
DSS Import FillOption= 0

--- K120-00-00.g01 (geometry) ---

Geom Title=K120-00-00 June 2007
Version=Version 3.0.1  Mar 2001

River Reach=K120-00-00      ,K120-00-00_0022
Reach XY= 30
      3100554.43     13955996.16      3100511.46     13955707.43
       3100636.6     13955219.71      3100375.99     13954257.78
      3100550.47     13953631.91      3100314.25     13953398.08
      3100101.57     13952621.17      3100236.12     13951694.52
      3100161.25     13951490.53      3100573.58     13950652.86
       3100586.6     13950248.12      3101061.86     13949188.01
      3100958.78     13948851.64      3100565.98     13948495.74
      3100868.72     13948104.03      3100963.66     13947725.66
      3100930.57     13946898.52        3101077.       13946574.
      3100994.59     13944603.59      3101281.04      13944370.3
      3101617.41     13944374.64        3101922.       13944242.
      3102216.26     13943607.61       3102465.4     13943439.21
      3102585.02     13943190.92      3102286.58     13942816.81
      3102044.39     13942793.37      3101938.49     13942552.05
      3101915.92     13942440.94      3102162.45      13942126.7

Type RM Length L Ch R = 1 ,16297.90,538,565.9,588
BEGIN DESCRIPTION:
Cross Section K120-00-00-X08
END DESCRIPTION:
XS GIS Cut Line= 4
      3101363.51      13956034.4      3100611.11     13955975.53
      3100502.68     13956007.33      3099671.82      13956353.1
#Sta/Elev= 30
  4184.1  117.72    4231   118.1  4612.2  115.52    4701   114.9    4711   115.3
    4751   112.6    4771     114    4911   115.9  4911.9  115.39  4933.6  114.78
  4955.2  113.12  4978.4     113  4994.2  108.02  4995.6   107.2  4996.6  105.84
  4999.1  105.38  5002.8  106.03  5006.1  107.85  5013.5  108.85  5025.7  113.32
  5045.2  112.34  5060.4  116.51  5073.5   116.4  5101.8   117.6  5161.8   117.5
  5211.8   113.9  5241.8   113.8  5321.8   114.4  5391.8   116.7  5951.8   119.3
#Mann= 6 ,-1 , 0
  4184.1     .09       0  4612.2     .06       0  4955.2    .045       0
  4978.4     .04       0  5025.7    .045       0  5045.2     .99       0
Bank Sta=4978.4,5025.7
XS Rating Curve= 0
Exp/Cntr=.3,.1

Type RM Length L Ch R = 1 ,15732.  ,101,99.1,96
BEGIN DESCRIPTION:
interpolated channel - LIDAR overbanks
WOOD BRIDGE 350' US LOUETTA - XS4
END DESCRIPTION:
XS GIS Cut Line= 5
      3101436.46     13955871.98      3100628.93     13955464.83
      3100551.97     13955422.63      3100456.94     13955383.24
      3099813.19     13955528.91
#Sta/Elev= 30
    4061   118.1    4111   118.2    4151  117.45    4161  116.37    4181  117.55
    4261  116.56    4291  117.09    4351  116.48    4361  115.62    4501  115.62
    4561  114.09    4641  113.21    4811  112.77    4831   112.2    4851  112.65
  4965.4   112.3 4989.64   108.9 4993.28   105.9 4999.87  104.13 5006.53   105.8
 5008.08  107.12 5012.95  108.54  5035.4  111.49    5186  111.62    5226  114.55
    5256  114.86    5306  112.98    5476  114.41    5516  115.32    5816  116.44
#Mann= 3 ,-1 , 0
    4061     .09       0  4965.4    .055       0  5035.4      .1       0
Bank Sta=4965.4,5035.4
XS Rating Curve= 0
Exp/Cntr=.5,.3

Type RM Length L Ch R = 1 ,15632.90,40.2,40.2,40.2
BEGIN DESCRIPTION:
Upstream Section of Bridge/Culvert/Weir
WOOD BRIDGE 350' US LOUETTA - XS 3
END DESCRIPTION:
XS GIS Cut Line= 5
      3101473.46      13955786.4      3100655.57     13955363.86
      3100601.72     13955343.67      3100493.95     13955297.66
       3099850.2      13955443.3
#Sta/Elev= 30
  4060.7  117.72  4140.7  117.72  4387.7  115.56  4450.7  115.02  4510.7  115.32
  4530.7  114.72  4540.7  115.02  4670.7  113.02  4710.7  113.42  4785.6  112.23
  4937.1  111.34  4990.5  112.14  4991.3  108.28  4994.4  105.12    5000  103.91
  5005.6   105.3  5006.9  106.74    5011   107.8  5011.7  111.03  5068.5   109.6
  5121.3  110.72  5225.9  111.37    5246  112.02    5266  113.72    5296  114.82
    5346  113.02    5486  114.62    5546  114.92    5566  115.72    5816  116.22
#Mann= 4 ,-1 , 0
  4060.7     .06       0  4387.7     .09       0  4990.5    .055       0
  5011.7      .1       0
#XS Ineff= 2 , 0
       0    4970  111.58    5030       0  110.28
Permanent Ineff=
       F       F
Bank Sta=4990.5,5011.7
XS Rating Curve= 0
Exp/Cntr=.5,.3

Type RM Length L Ch R = 3 ,15612.80,,,
BEGIN DESCRIPTION:
WOOD BRIDGE 350' US LOUETTA
Structure ID: K120-00-00-S4-1
END DESCRIPTION:
Bridge Culvert--1,0,-1,-1, 0
Deck Dist Width WeirC Skew NumUp NumDn MinLoCord MaxHiCord MaxSubmerge Is_Ogee
10,15,2.6,0, 42, 42, , , .95, 0, ,,,
  4060.7  4070.7  4090.7  4140.7  4210.7  4230.7  4240.7  4450.7  4510.7  4530.7
  4540.7  4670.7  4710.7  4785.6  4835.7    4892  4937.1  4949.9  4990.5  4991.3
 4991.51  4991.6  5002.7 5011.29  5011.4  5011.7  5014.9  5067.3  5068.5  5121.3
    5172  5225.9    5246    5266    5296    5316    5326    5346    5486    5546
    5566    5816
   117.7   117.8   117.5   117.7   116.9   117.1   116.8     115   115.3   114.7
     115     113   113.4  112.21  112.11  111.72  111.59  111.58  112.13  111.98
  111.98  111.98  111.89  111.91  111.91  111.89  111.72  110.28  110.29  110.77
   111.2  111.82     112   113.7   114.8   114.2   113.5     113   114.6   114.9
   115.7   116.2
   117.7   117.8   117.5   117.7   116.9   117.1   116.8     115   115.3   114.7
     115     113   113.4  112.21  112.11  111.71  111.32  111.51  112.12  108.26
  108.01  110.78  110.69  110.71  109.63  111.01  110.93  109.61  109.58   110.7
  111.15  111.35     112   113.7   114.8   114.2   113.5     113   114.6   114.9
   115.7   116.2
  4060.7  4070.7  4090.7  4140.7  4210.7  4230.7  4240.7  4450.7  4510.7  4530.7
  4540.7  4670.7  4710.7  4785.6  4835.7    4892  4937.1  4949.9  4990.5  4991.3
 4991.51  4991.6  5002.7 5011.29  5011.4  5011.7  5014.9  5067.3  5068.5  5121.3
    5172  5225.9    5246    5266    5296    5316    5326    5346    5486    5546
    5566    5816
   117.7   117.8   117.5   117.7   116.9   117.1   116.8     115   115.3   114.7
     115     113   113.4  112.21  112.11  111.72  111.59  111.58  112.13  111.98
  111.98  111.98  111.89  111.91  111.91  111.89  111.72  110.28  110.29  110.77
   111.2  111.82     112   113.7   114.8   114.2   113.5     113   114.6   114.9
   115.7   116.2
   117.7   117.8   117.5   117.7   116.9   117.1   116.8     115   115.3   114.7
     115     113   113.4  112.21  112.11  111.71  111.32  111.51  112.12  108.26
  108.01  110.78  110.69  110.71  109.63  111.01  110.93  109.61  109.58   110.7
  111.15  111.35     112   113.7   114.8   114.2   113.5     113   114.6   114.9
   115.7   116.2
BR Coef= 1 , 0 , 0 ,1.25, 0 ,,,.8,0,2,0,
WSPro=,,,, 1 ,,,, 0 ,,,, 0 ,,,,-1 ,-1 ,-1 , 0 , 0 , 0 , 0 , 0
BR U #Sta/Elev= 62
  4060.7   117.7  4070.7   117.8  4090.7   117.5  4140.7   117.7  4210.7   116.9
  4230.7   117.1  4240.7   116.8  4387.7  115.54  4450.7     115  4510.7   115.3
  4530.7   114.7  4540.7     115  4670.7     113  4710.7   113.4  4785.6  112.21
    4790  112.25  4835.7  112.11  4841.8  112.07  4887.5  111.75    4892  111.71
  4937.1  111.32  4949.9  111.51  4990.5  112.12  4991.3  108.26  4991.4  108.14
 4991.51  108.01  4991.6  107.91  4991.7  107.79  4992.6  106.73  4994.3  105.38
  4994.4   105.1    5000  103.89  5002.7  104.56  5005.6  105.28  5005.7  105.47
  5006.9  106.72    5011  107.78  5011.2   108.7 5011.29  109.12  5011.4  109.63
  5011.5  110.09  5011.7  111.01  5014.9  110.93  5067.3  109.61  5068.5  109.58
  5118.6  110.64  5121.3   110.7    5172  111.15  5172.1  111.15  5222.2  111.35
  5225.9  111.35  5232.9  111.58    5246     112    5266   113.7    5296   114.8
    5316   114.2    5326   113.5    5346     113    5486   114.6    5546   114.9
    5566   115.7    5816   116.2
BR U #Mann= 4
  4060.7     .06  4387.7     .09  4990.5    .055  5011.7      .1
BR D #Sta/Elev= 62
  4060.7   117.7  4070.7   117.8  4090.7   117.5  4140.7   117.7  4210.7   116.9
  4230.7   117.1  4240.7   116.8  4387.7  115.54  4450.7     115  4510.7   115.3
  4530.7   114.7  4540.7     115  4670.7     113  4710.7   113.4  4785.6  112.21
    4790  112.25  4835.7  112.11  4841.8  112.07  4887.5  111.75    4892  111.71
  4937.1  111.32  4949.9  111.51  4990.5  112.12  4991.3  108.26  4991.4  108.14
 4991.51  108.01  4991.6  107.91  4991.7  107.79  4992.6  106.73  4994.3  105.38
  4994.4   105.1    5000  103.89  5002.7  104.56  5005.6  105.28  5005.7  105.47
  5006.9  106.72    5011  107.78  5011.2   108.7 5011.29  109.12  5011.4  109.63
  5011.5  110.09  5011.7  111.01  5014.9  110.93  5067.3  109.61  5068.5  109.58
  5118.6  110.64  5121.3   110.7    5172  111.15  5172.1  111.15  5222.2  111.35
  5225.9  111.35  5232.9  111.58    5246     112    5266   113.7    5296   114.8
    5316   114.2    5326   113.5    5346     113    5486   114.6    5546   114.9
    5566   115.7    5816   116.2
BR D #Mann= 4
  4060.7     .06  4387.7     .09  4990.5    .055  5011.7      .1
BC Design=,, 0 ,, 0 ,,,,,,
BC HTab HWMax=117.82

Type RM Length L Ch R = 1 ,15592.70,124,108.7,84
BEGIN DESCRIPTION:
Downstream Section of Bridge/Culvert/Weir
WOOD BRIDGE 350' US LOUETTA - XS 2
END DESCRIPTION:
XS GIS Cut Line= 5
      3101483.37       13955749.      3100664.42     13955325.93
      3100609.88     13955305.48      3100496.58     13955257.11
      3099846.51      13955404.2
#Sta/Elev= 30
  4060.7  117.67  4140.7  117.67  4387.7  115.51  4450.7  114.97  4510.7  115.27
  4530.7  114.67  4540.7  114.97  4670.7  112.97  4710.7  113.37  4785.6  112.18
  4937.1  111.29  4990.5  112.09  4991.3  108.23  4994.4  105.07    5000  103.86
  5005.6  105.25  5006.9  106.69    5011  107.75  5011.7  110.98  5068.5  109.55
  5121.3  110.67  5225.9  111.32    5246  111.97    5266  113.67    5296  114.77
    5346  112.97    5486  114.57    5546  114.87    5566  115.67    5816  116.17
#Mann= 4 ,-1 , 0
  4060.7     .06       0  4387.7     .09       0  4990.5    .055       0
  5011.7      .1       0
#XS Ineff= 2 , 0
       0 4983.83  111.58 5018.37       0  110.28
Permanent Ineff=
       F       F
Bank Sta=4990.5,5011.7
XS Rating Curve= 0
Exp/Cntr=.5,.3

Type RM Length L Ch R = 1 ,15484.  ,124.6,123,107.7
BEGIN DESCRIPTION:
interpolated channel - LIDAR overbanks
WOOD BRIDGE 350' US LOUETTA - XS 1
END DESCRIPTION:
XS GIS Cut Line= 4
      3101476.43     13955647.25      3100684.62     13955204.32
      3100547.12     13955219.23      3099821.52     13955379.92
#Sta/Elev= 30
  4042.6  116.72  4172.6  116.18  4252.6  116.65  4362.6  115.81  4392.6  114.94
  4552.6  113.46  4722.6  113.24  4752.6  114.11  4812.6  114.66  4832.6   114.2
  4852.6  113.06  4959.9  111.88 4977.95  108.65 4985.17  105.59 4987.75  105.04
 4999.17  103.84 5009.71  105.56 5011.73  106.83  5029.9  109.07  5039.9  110.09
  5059.9  110.89  5248.2  112.15  5268.2     114  5298.2  114.74  5328.2  113.66
  5378.2  113.04  5468.2  114.52  5528.2  114.71  5548.2  115.43  5831.4  116.27
#Mann= 3 ,-1 , 0
  4042.6     .09       0  4959.9     .04       0  5059.9      .1       0
Bank Sta=4959.9,5059.9
XS Rating Curve= 0
Exp/Cntr=.3,.1

Type RM Length L Ch R = 1 ,15361.  ,85,97.1,101
BEGIN DESCRIPTION:
interpolated channel - LIDAR overbanks
LOUETTA - XS 4
END DESCRIPTION:
XS GIS Cut Line= 4
      3101488.37     13955526.81      3100676.34     13955083.39
      3100535.53     13955094.98      3099761.58     13955323.03
#Sta/Elev= 30
  4013.1  116.21  4223.1  116.53  4633.1  113.09  4653.1  113.48  4713.1  113.28
  4843.1  111.51  4923.1  112.49  4958.3  111.42  4968.3  110.36 4989.06  105.25
 5006.64   104.6 5008.24  103.82 5012.11  103.82 5016.35  104.94 5023.93  105.81
  5027.2     107  5028.3   108.4  5048.3  110.23  5078.3  110.83  5119.6  110.64
  5229.6  112.29  5279.6   114.7  5339.6  114.74  5359.6  113.58  5369.6  114.15
  5389.6  114.26  5439.6  113.43  5499.6  114.71  5679.6  116.35  5886.4  116.11
#Mann= 3 ,-1 , 0
  4013.1     .09       0  4958.3     .04       0  5048.3      .1       0
Bank Sta=4958.3,5048.3
XS Rating Curve= 0
Exp/Cntr=.5,.3

Type RM Length L Ch R = 1 ,15263.90,100.3,100.3,100.3
BEGIN DESCRIPTION:
Upstream Section of Bridge/Culvert/Weir Louetta
LOUETTA - XS 3
END DESCRIPTION:
XS GIS Cut Line= 4
      3101467.55      13955429.6      3100669.85     13955000.75
      3100494.23     13954988.57      3099740.76      13955225.8
#Sta/Elev= 30
  4018.6  116.13  4128.6  116.73  4238.6  116.53  4548.6  113.13  4668.6  113.53
  4738.6  112.43  4748.7  111.42  4779.7  111.07  4848.7  111.61 4939.81  111.22
  4944.9   111.2  4972.3   105.4  4995.4  104.87  4997.5  103.81    5003  103.81
  5008.2  105.19  5017.5  106.06  5034.4  110.54  5042.5  110.48  5086.5  110.14
  5270.2  111.16  5276.6  113.91  5290.3  114.53  5360.3  114.63  5380.3  113.83
  5500.3  114.23  5690.3  116.23  5820.3  116.43  5870.3  115.63  5890.3  116.63
#Mann= 8 ,-1 , 0
  4018.6     .06       0  4128.6     .08       0 4939.81    .045       0
  4944.9    .055       0  5034.4    .045       0  5042.5     .07       0
  5270.2     .06       0  5380.3      .1       0
#XS Ineff= 2 , 0
       0  4934.9   113.1  5044.4       0  113.53
Permanent Ineff=
       F       F
Bank Sta=4944.9,5034.4
XS Rating Curve= 0
Exp/Cntr=.5,.3

Type RM Length L Ch R = 3 ,15213.75,,,
BEGIN DESCRIPTION:
LOUETTA
Structure ID: K120-00-00-S4
END DESCRIPTION:
Bridge Culvert--1,0,-1,-1, 0
Deck Dist Width WeirC Skew NumUp NumDn MinLoCord MaxHiCord MaxSubmerge Is_Ogee
10,83,2.6,0, 48, 48, , , .95, 0, ,,,
  4018.6  4048.6  4128.6  4138.6  4238.6  4258.6  4548.6  4618.8    4668  4668.6
  4738.6  4748.7  4779.7  4811.8 4816.69    4855 4855.01    4940 4940.01    5034
 5034.01    5065 5065.01    5140 5140.01    5145  5147.6  5190.4  5198.9  5252.4
  5270.2  5272.9  5276.6  5280.3  5290.3  5360.3  5380.3  5500.3  5530.3  5540.3
  5650.3  5670.3  5690.3  5700.3  5820.3  5850.3  5870.3  5890.3
   116.1   116.7   116.7   116.4   116.5   115.9   113.1  113.33   113.5   113.5
  113.53  113.54  113.55  113.57  113.58  113.58  115.07  115.94   117.2   117.3
   117.3   117.3  115.94  115.19  113.55  113.55  113.55  113.61  113.64  113.83
  113.89   113.9  113.88     114   114.5   114.6   113.8   114.2   114.7   114.6
     116   115.8   116.2     116   116.4   115.5   115.6   116.6
   116.1   116.7   116.7   116.4   116.5   115.9   113.1  113.33   113.5   113.5
   112.4  111.39  111.04  111.29  111.33  110.84  110.84  110.84  110.84  110.84
     110     110     110     110     110     110  110.39  110.64  110.69  110.85
  111.13  112.29  113.88     114   114.5   114.6   113.8   114.2   114.7   114.6
     116   115.8   116.2     116   116.4   115.5   115.6   116.6
  4018.6  4048.6  4128.6  4138.6  4238.6  4258.6  4548.6  4618.8    4668  4668.6
  4738.6  4748.7  4779.7  4811.8 4816.69    4855 4855.01    4940 4940.01    5034
 5034.01    5065 5065.01    5140 5140.01    5145  5147.6  5190.4  5198.9  5252.4
  5270.2  5272.9  5276.6  5280.3  5290.3  5360.3  5380.3  5500.3  5530.3  5540.3
  5650.3  5670.3  5690.3  5700.3  5820.3  5850.3  5870.3  5890.3
   116.1   116.7   116.7   116.4   116.5   115.9   113.1  113.33   113.5   113.5
  113.53  113.54  113.55  113.57  113.58  113.58  115.07  115.94   117.2   117.3
   117.3   117.3  115.94  115.19  113.55  113.55  113.55  113.61  113.64  113.83
  113.89   113.9  113.88     114   114.5   114.6   113.8   114.2   114.7   114.6
     116   115.8   116.2     116   116.4   115.5   115.6   116.6
   116.1   116.7   116.7   116.4   116.5   115.9   113.1  113.33   113.5   113.5
   112.4  111.39  111.04  111.29  111.33  110.83  110.83  110.83  110.83  110.83
     110     110     110     110     110     110  110.39  110.64  110.69  110.85
  111.13  112.29  113.88     114   114.5   114.6   113.8   114.2   114.7   114.6
     116   115.8   116.2     116   116.4   115.5   115.6   116.6
Pier Skew, UpSta & Num, DnSta & Num=  ,4977.2, 2 ,4977.2, 2 , 0 , 0 , 0 ,,
     1.3     1.3
  104.32  112.71
     1.3     1.3
   105.2  113.59
Pier Skew, UpSta & Num, DnSta & Num=  ,5008.6, 2 ,5008.6, 2 , 0 , 0 , 0 ,,
     1.3     1.3
  104.09  112.68
     1.3     1.3
  104.97  113.56
BR Coef= 1 , 1 , 1 ,1.25, 0 ,,,.8,0,2,0,
WSPro=,,,, 1 ,,,, 0 ,,,, 0 ,,,,-1 ,-1 ,-1 , 0 , 0 , 0 , 0 , 0
BR U #Sta/Elev= 71
  4018.6  116.13  4048.6  116.73  4128.6  116.73  4138.6  116.43  4238.6  116.53
  4258.6  115.93  4548.6  113.13  4618.8  113.36    4668  113.53  4668.6  113.53
  4738.6  112.43  4748.7  111.42  4779.7  111.07  4811.8  111.32 4816.69  111.36
  4816.8  111.36 4816.91  111.36  4848.7  111.61  4866.1  111.54  4903.2  111.38
 4939.81  111.22  4939.9  111.22  4944.9   111.2  4956.4  108.77  4972.2  105.42
  4972.3   105.4  4975.7  105.41  4989.3  105.04  4995.4  104.87  4996.6  103.84
  4997.5  103.81    4999  103.81    5003  103.81  5003.4  103.87  5008.2  105.19
  5008.6  105.23  5017.4  106.05  5017.5  106.06  5034.4  110.54 5039.39   110.5
  5039.5   110.5  5042.5  110.48  5086.5  110.14  5097.2  110.19 5129.79  110.34
  5129.9  110.34 5130.01  110.34  5133.8  110.36    5145  110.41  5147.6  110.42
  5190.4  110.67  5198.9  110.72  5252.4  110.88  5270.2  111.16  5272.9  112.32
  5276.6  113.91  5280.3  114.03  5290.3  114.53  5360.3  114.63  5380.3  113.83
  5500.3  114.23  5530.3  114.73  5540.3  114.63  5650.3  116.03  5670.3  115.83
  5690.3  116.23  5700.3  116.03  5820.3  116.43  5850.3  115.53  5870.3  115.63
  5890.3  116.63
BR U #Mann= 10
  4018.6     .06  4128.6     .08 4939.81    .045  4944.9    .025  4975.7     .04
  5008.6    .025  5034.4    .045  5042.5     .07  5270.2     .06  5380.3      .1
BR U Banks=4944.9,5034.4
BR D #Sta/Elev= 71
  4018.6  116.13  4048.6  116.73  4128.6  116.73  4138.6  116.43  4238.6  116.53
  4258.6  115.93  4548.6  113.13  4618.8  113.36    4668  113.53  4668.6  113.53
  4738.6  112.43  4748.7  111.42  4779.7  111.07  4811.8  111.32 4816.69  111.36
  4816.8  111.36 4816.91  111.36  4848.7  111.61  4866.1  111.54  4903.2  111.38
 4939.81  111.22  4939.9  111.22  4944.9   111.2  4956.4  108.62  4972.2  105.27
  4972.3  105.25  4975.7  105.26  4989.3  104.89  4995.4  104.72  4996.6  103.69
  4997.5  103.66    4999  103.66    5003  103.66  5003.4  103.72  5008.2  105.04
  5008.6  105.08  5017.4   105.9  5017.5  105.91  5034.4  110.54 5039.39   110.5
  5039.5   110.5  5042.5  110.48  5086.5  110.14  5097.2  110.19 5129.79  110.34
  5129.9  110.34 5130.01  110.34  5133.8  110.36    5145  110.41  5147.6  110.42
  5190.4  110.67  5198.9  110.72  5252.4  110.88  5270.2  111.16  5272.9  112.32
  5276.6  113.91  5280.3  114.03  5290.3  114.53  5360.3  114.63  5380.3  113.83
  5500.3  114.23  5530.3  114.73  5540.3  114.63  5650.3  116.03  5670.3  115.83
  5690.3  116.23  5700.3  116.03  5820.3  116.43  5850.3  115.53  5870.3  115.63
  5890.3  116.63
BR D #Mann= 10
  4018.6     .06  4128.6     .08 4939.81    .045  4944.9    .025  4975.7     .04
  5008.6    .025  5034.4    .045  5042.5     .07  5270.2     .06  5380.3      .1
BR D Banks=4944.9,5034.4
BC Design=,, 0 ,, 0 ,,,,,,
BC HTab HWMax=116.73

Type RM Length L Ch R = 1 ,15163.60,118,103.6,88
BEGIN DESCRIPTION:
Downstream Section of Bridge/Culvert/Weir  Louetta
LOUETTA - XS 2
END DESCRIPTION:
XS GIS Cut Line= 4
      3101463.94      13955333.5      3100662.45     13954902.63
      3100478.76     13954889.89      3099721.68      13955128.3
#Sta/Elev= 30
  4018.6  116.13  4128.6  116.73  4238.6  116.53  4548.6  113.13  4668.6  113.53
  4738.6  112.43  4748.7  111.42  4779.7  111.07  4848.7  111.61 4939.81  111.22
  4944.9   111.2  4972.3  105.25  4995.4  104.72  4997.5  103.66    5003  103.66
  5008.2  105.04  5017.5  105.91  5034.4  110.54  5042.5  110.48  5086.5  110.14
  5270.2  111.16  5276.6  113.91  5290.3  114.53  5360.3  114.63  5380.3  113.83
  5500.3  114.23  5690.3  116.23  5820.3  116.43  5870.3  115.63  5890.3  116.63
#Mann= 8 ,-1 , 0
  4018.6     .06       0  4128.6     .08       0 4939.81    .045       0
  4944.9     .04       0  5034.4    .045       0  5042.5     .07       0
  5270.2     .06       0  5380.3      .1       0
#XS Ineff= 2 , 0
       0 4938.23   113.1 5041.07       0  113.53
Permanent Ineff=
       F       F
Bank Sta=4944.9,5034.4
XS Rating Curve= 0
Exp/Cntr=.5,.3

Type RM Length L Ch R = 1 ,15060.  ,1409,1383.4,1326
BEGIN DESCRIPTION:
interpolated channel - LIDAR overbanks
LOUETTA - XS 1
END DESCRIPTION:
XS GIS Cut Line= 4
      3101445.44     13955241.07       3100616.7     13954780.22
      3100507.29     13954806.97      3099703.18     13955035.83
#Sta/Elev= 30
    3989  118.15    4069  120.08    4109  120.01    4139  119.74    4209   117.7
    4309  115.68    4559  113.03    4599  113.55    4609  113.12    4669  112.66
    4699  111.45    4859  110.91    4919  111.71  4937.3   111.4  4967.3   109.8
  4977.3  108.34 4986.59  105.08 5005.79  104.13 5006.96  103.17 5007.84  103.14
 5012.96  103.14 5018.24  104.84 5027.58  105.88  5037.3  109.54  5049.9  110.78
  5099.9  110.35  5219.9  110.83  5299.9  114.03  5549.9   115.7  5885.9  117.25
#Mann= 5 ,-1 , 0
    3989     .08       0    4559     .14       0  4967.3     .04       0
  5049.9     .12       0  5219.9     .08       0
Bank Sta=4967.3,5049.9
XS Rating Curve= 0
Exp/Cntr=.3,.1

Type RM Length L Ch R = 1 ,13676.60,293,346.6,389
BEGIN DESCRIPTION:
Cross Section K120-00-00-X7
END DESCRIPTION:
XS GIS Cut Line= 4
      3101398.79      13953357.5      3100460.06     13953489.88
      3100436.72     13953634.88      3099775.48      13954274.5
#Sta/Elev= 30
  3981.4   113.5  4471.4   110.5  4501.4   109.7  4541.4   110.2  4741.4     108
  4751.4   108.7  4859.7  107.56  4935.1  104.96  4968.7  106.69  4992.4  101.92
  4997.5    96.6  5002.4   96.15  5003.8   97.54  5005.3  101.15  5026.1  107.45
  5040.6  110.02  5100.1   107.5  5186.3   109.2  5196.3   108.2  5456.3   109.6
  5496.3   109.2  5536.3   110.3  5586.3   109.5  5686.3   110.9  5726.3   109.8
  5776.3   110.7  5816.3   110.5  5876.3   112.5  5936.3   111.6  5996.3   113.2
#Mann= 3 ,-1 , 0
  3981.4     .14       0  4968.7     .08       0  5040.6     .14       0
Bank Sta=4968.7,5040.6
XS Rating Curve= 0
Exp/Cntr=.3,.1

Type RM Length L Ch R = 1 ,13330.  ,97,96.4,95
BEGIN DESCRIPTION:
interpolated channel - LIDAR overbanks
SHEET PILING DROP STRUCTURE 45' US OF LEXINGTON RD - XS 4
END DESCRIPTION:
XS GIS Cut Line= 4
      3101487.49     13953036.38       3100339.5      13953259.9
      3100228.92     13953294.45      3099602.78     13953954.76
#Sta/Elev= 30
  3782.7  113.63  3832.7  114.21  3962.7  113.76  4222.7  111.72  4252.7  110.86
  4412.7  109.97  4492.7  110.32  4642.7  108.08  4832.7  107.74  4872.7  106.31
  4902.7  107.31  4942.7   106.3  4962.2  104.52  4982.2  100.06 4989.17    99.4
 4990.51   97.28 4991.85   96.77 4997.32   96.55 5000.35   98.11  5022.2  103.59
  5042.2  106.72  5468.1  109.04  5488.1  108.41  5558.1  109.27  5668.1  109.06
  5738.1  110.96  5878.1  112.21  5928.1  111.29  5948.1  110.07  5978.1  110.22
#Mann= 4 ,-1 , 0
  3782.7     .14       0  4942.7    .045       0  5042.2     .14       0
  5488.1      .1       0
Bank Sta=4942.7,5042.2
XS Rating Curve= 0
Exp/Cntr=.7,.5

Type RM Length L Ch R = 1 ,13233.60,20,20,20
BEGIN DESCRIPTION:
Upstream Section of Bridge/Culvert/Weir
SHEET PILING DROP STRUCTURE 45' US OF LEXINGTON RD - XS 3
END DESCRIPTION:
XS GIS Cut Line= 4
      3101462.04      13952943.8      3100314.06     13953167.38
      3100203.47     13953201.94      3099577.33      13953862.2
#Sta/Elev= 30
  3785.9  113.99  4405.9  109.89  4425.9  109.29  4495.9  110.39  4525.9  109.79
  4565.9  109.89  4605.9  108.29  4795.9  108.19    4944  105.67  4960.9  105.82
  4993.9   99.56  4995.2   97.21  4996.6   96.83  5002.3   96.66  5033.8  104.07
  5042.6  106.17  5042.7  105.96  5057.4  105.95  5076.6  106.68  5241.3  108.19
  5261.3  107.59  5281.3  107.99  5321.3  107.19  5461.3  108.79  5551.3  108.09
  5651.3  110.69  5661.3  111.19  5851.3  111.79  5891.3  110.39  5981.3  112.69
#Mann= 5 ,-1 , 0
  3785.9     .14       0  4960.9     .02       0  5033.8    .045       0
  5076.6     .12       0  5281.3      .1       0
#XS Ineff= 2 , 0
       0    4984   103.6    5016       0   103.6
Permanent Ineff=
       F       F
Bank Sta=4960.9,5042.7
XS Rating Curve= 0
Exp/Cntr=.7,.5

Type RM Length L Ch R = 5 ,13223.60,,,
BEGIN DESCRIPTION:
SHEET PILING DROP STRUCTURE 45' US OF LEXINGTON RD.
***SEE NOTES BELOW***
***U/S N VALUE IS 0.06.  D/S N IS O.O3***
Structure ID: K120-00-00-S3b
END DESCRIPTION:
IW Pilot Flow=0
#Inline Weir SE= 30
  2465.9   119.6  2605.9   114.8  2845.9   116.4  3055.9   114.5  3245.9   116.9
  4795.9   108.2  4960.9  105.84  4993.8  103.63    4994   99.57  4996.7   99.61
  4996.9    96.8  5002.3   96.68  5003.2   96.76  5003.5   99.64    5006   99.63
  5006.1  103.66  5042.6  106.19  5241.3   108.2  5551.3   108.1  5661.3   111.2
  5891.3   110.4  5981.3   112.7  6111.3   110.3  6151.3   112.9  6561.3   113.7
  6621.3   117.2  6711.3     114  6831.3   116.8  6871.3   115.2  7881.4   120.3
IW Dist,WD,Coef,Skew,MaxSub,Min_El,Is_Ogee,SpillHt,DesHd
10,1,3,0,.95,, 0 ,,,0,0,

Type RM Length L Ch R = 1 ,13213.60,28,28.1,28.1
BEGIN DESCRIPTION:
Cross Section FIELD_DS
SHEET PILING DROP STRUCTURE 45' US OF LEXINGTON RD - XS 2
LEXINGTON RD. - XS 4
***SEE NOTES BELOW***
***U/S N VALUE IS 0.06.  D/S N IS O.O3***
Located At: SHEET PILING DROP STRUCTURE 45' US OF LEXINGTON RD.
END DESCRIPTION:
XS GIS Cut Line= 5
      3101422.43      13952929.2      3100286.29     13953155.13
      3100232.97      13953171.9      3100183.73     13953187.13
      3099592.88      13953811.9
#Sta/Elev= 28
    3820  113.78    4400  109.93    4430  109.54    4470  110.37    4570  109.86
    4610  108.52    4790     108    4880  106.72    4890  106.81    4950  105.68
  4959.9  105.86    4960  105.86  4996.6   93.93  5003.4   93.86  5042.8  105.97
  5044.3  105.01  5064.3  105.71  5074.3  106.47  5085.8  106.81  5205.8  107.52
  5245.8  107.02  5295.8  107.03  5405.8  108.49  5525.8  108.27  5575.8  110.11
  5815.8   111.9  5885.8  110.23  5945.8  110.98
#Mann= 5 ,-1 , 0
    3820     .14       0  4959.9     .02       0  5042.8    .045       0
  5074.3     .12       0  5295.8      .1       0
Bank Sta=4959.9,5042.8
XS Rating Curve= 0
Exp/Cntr=.7,.5

Type RM Length L Ch R = 1 ,13185.50,254.8,254.8,254.8
BEGIN DESCRIPTION:
Upstream Section of Bridge/Culvert/Weir
LEXINGTON RD. - XS 3
END DESCRIPTION:
XS GIS Cut Line= 4
       3101079.3      13952968.7      3100295.09     13953122.64
      3100177.01     13953160.32      3099582.35      13953795.4
#Sta/Elev= 30
  4160.6  112.03  4180.6  111.23  4270.6  111.43  4290.6  110.73  4440.6  109.53
  4590.6  109.33  4653.1  106.88  4926.5  106.95 4972.79  105.85  4973.9  105.83
  4989.8   96.46  4991.9   93.87  5006.7   93.74  5009.1   94.97  5010.2   96.26
  5031.7   95.92  5065.2  107.03  5168.9  107.99  5183.7  106.83  5203.7  106.63
  5263.7  107.13  5333.7  108.33  5433.7  107.53  5483.7  107.93  5523.7  109.23
  5593.7  110.63  5773.7  111.03  5813.7  111.73  5873.7  110.23  5953.7  110.73
#Mann= 6 ,-1 , 0
  4160.6     .14       0  4926.5    .045       0 4972.79     .02       0
  5031.7    .045       0  5065.2     .06       0  5483.7      .1       0
#XS Ineff= 2 , 0
       0  4963.9  106.43  5075.2       0   107.1
Permanent Ineff=
       F       F
Bank Sta=4973.9,5065.2
XS Rating Curve= 0
Exp/Cntr=.5,.3

Type RM Length L Ch R = 2 ,13058.10,,,
BEGIN DESCRIPTION:
LEXINGTON RD.  field surveyed negative culvert slope
 ***SEE NOTES BELOW***
***D/S N VALUE SHOULD BE 0.04***
***U/S N VALUE SHOULD BE 0.03***
***U/S XS SHOULD MATCH D/S XS OF WEIR***
***MAKE CHANGES IN RAS***
Structure ID: K120-00-00-S3a
END DESCRIPTION:
Bridge Culvert--1,0,-1,-1, 0
Deck Dist Width WeirC Skew NumUp NumDn MinLoCord MaxHiCord MaxSubmerge Is_Ogee
10,236,3,0, 60, 60, , , .95, 0, ,,,
  2430.6  2480.6  2500.6  2520.6  2550.6  2580.6  3130.6  3160.6  3200.6  3370.6
  3520.6  3550.6  3640.6  3680.6  3710.6  3780.6  3810.6  3890.6  3980.6  4440.6
  4590.6  4653.1  4926.5  4973.9  4989.8  4991.9  5006.7  5010.2  5031.7  5065.2
  5101.6  5168.9  5203.7  5263.7  5333.7  5433.7  5593.7  5813.7  5873.7  5953.7
  6023.7  6093.7  6133.7  6183.7  6363.7  6553.7  6603.7  6633.7  6663.7  6703.7
  6733.7  6773.7  6803.7  6843.7  6863.7  6883.7  6903.7  6923.7  7173.7  7938.3
   119.4   119.7   118.6   115.8   115.7   114.2     116   116.9   115.6   115.2
   116.4   115.2     115   115.9   114.8   115.1   114.1   114.6   112.5   109.5
   109.3  106.85  106.93   107.7  107.83  107.84  107.91  107.91  107.44  107.54
  107.72  107.97  107.26  107.13   108.3   107.5   110.6   111.7   110.2   110.7
   112.7   110.7   110.7   113.2   113.4     115   113.8   116.6   117.2   116.3
   113.9   115.6   115.6   117.5   115.9   116.2     115     116   117.6   120.3
   119.4   119.7   118.6   115.8   115.7   114.2     116   116.9   115.6   115.2
   116.4   115.2     115   115.9   114.8   115.1   114.1   114.6   112.5   109.5
   109.3  106.85  106.92   105.8   96.43   93.84   93.71   96.23   95.89     107
  107.58  107.96   106.6  107.13   108.3   107.5   110.6   111.7   110.2   110.7
   112.7   110.7   110.7   113.2   113.4     115   113.8   116.6   117.2   116.3
   113.9   115.6   115.6   117.5   115.9   116.2     115     116   117.6   120.3
  2430.6  2480.6  2500.6  2520.6  2550.6  2580.6  3130.6  3160.6  3200.6  3370.6
  3520.6  3550.6  3640.6  3680.6  3710.6  3780.6  3810.6  3890.6  3980.6  4440.6
  4590.6  4653.1  4926.5  4973.9  4989.8  4991.9  4999.1  5006.7  5010.2  5031.7
  5065.2  5168.9  5203.7  5263.7  5333.7  5483.7  5593.7  5813.7  5873.7  5953.7
  6023.7  6093.7  6133.7  6183.7  6363.7  6553.7  6603.7  6633.7  6663.7  6703.7
  6733.7  6773.7  6803.7  6843.7  6863.7  6883.7  6903.7  6923.7  7173.7  7938.3
  119.12  119.42  118.32  115.52  115.42  113.92  115.72  116.62  115.32  114.92
  116.12  114.92  114.72  115.62  114.52  114.82  113.82  114.32  112.22  109.22
  109.02  106.85  106.93   107.7  107.83  107.84   107.9  107.91  107.91  107.44
  107.54  107.97  107.26  106.82  108.02  107.62  110.32  111.42  109.92  110.42
  112.42  110.42  110.42  112.92  113.12  114.72  113.52  116.32  116.92  116.02
  113.62  115.32  115.32  117.22  115.62  115.92  114.72  115.72  117.32  120.02
  119.12  119.42  118.32  115.52  115.42  113.92  115.72  116.62  115.32  114.92
  116.12  114.92  114.72  115.62  114.52  114.82  113.82  114.32  112.22  109.22
  109.02  106.57  106.64  105.52   96.15   93.56   93.44   93.43   95.95   95.61
  106.72  107.68  106.32  106.82  108.02  107.62  110.32  111.42  109.92  110.42
  112.42  110.42  110.42  112.92  113.12  114.72  113.52  116.32  116.92  116.02
  113.62  115.32  115.32  117.22  115.62  115.92  114.72  115.72  117.32  120.02
BR Coef= 1 , 0 , 0 ,1.25, 0 ,,,.8,-1,2,0,
WSPro=,,,, 1 ,,,, 0 ,,,, 0 ,,,,-1 ,-1 ,-1 , 0 , 0 , 0 , 0 , 0
Culvert=2,8,14,236,.015,.4,1,8,1,93.66,4992.1,94.67,4992.1,Culvert #1  , 0 ,10
Culvert Bottom n=.015
Culvert=2,8,14,236,.015,.4,1,8,1,93.66,5007.1,94.67,5007.1,Culvert #2  , 0 ,10
Culvert Bottom n=.015
BC Design=,, 0 ,, 0 ,,,,,,
BC HTab HWMax=112.03

Type RM Length L Ch R = 1 ,12930.70,93,98.7,102
BEGIN DESCRIPTION:
Downstream Section of Bridge/Culvert/Weir
LEXINGTON RD. - XS 2
END DESCRIPTION:
XS GIS Cut Line= 4
      3101000.95      13952726.5      3100215.62     13952880.66
      3100091.48     13952920.27      3099493.26      13953559.1
#Sta/Elev= 30
  4160.6  111.72  4180.6  110.92  4270.6  111.12  4290.6  110.42  4440.6  109.22
  4590.6  109.02  4653.1  106.57  4926.5  106.64 4972.79  105.54  4973.9  105.52
  4989.8   96.15  4991.9   93.56  5006.7   93.43  5009.1   94.66  5010.2   95.95
  5031.7   95.61  5065.2  106.72  5168.9  107.68  5183.7  106.52  5203.7  106.32
  5263.7  106.82  5333.7  108.02  5433.7  107.22  5483.7  107.62  5523.7  108.92
  5593.7  110.32  5773.7  110.72  5813.7  111.42  5873.7  109.92  5953.7  110.42
#Mann= 6 ,-1 , 0
  4160.6     .14       0  4926.5    .045       0 4972.79     .04       0
  5031.7    .045       0  5065.2     .06       0  5483.7      .1       0
#XS Ineff= 2 , 0
       0 4967.23  106.12 5071.87       0  106.79
Permanent Ineff=
       F       F
Bank Sta=4973.9,5065.2
XS Rating Curve= 0
Exp/Cntr=.5,.3

Type RM Length L Ch R = 1 ,12832.  ,991,1049.4,1093
BEGIN DESCRIPTION:
interpolated channel - LIDAR overbanks
LEXINGTON RD. - XS 1
END DESCRIPTION:
XS GIS Cut Line= 4
       3100973.2     13952631.75      3100187.86     13952785.83
      3100063.73     13952825.44      3099465.51     13953464.34
#Sta/Elev= 30
  4157.9  111.38  4557.9   108.7  4707.9  105.96  4747.9  106.95  4797.9  105.56
  4847.9  106.57  4907.9  106.36  4937.9     106  4958.2  103.12 4968.89   96.25
 4971.02   93.84 4986.07   93.13 4989.48   95.47 5010.41   95.66 5026.95  101.12
  5028.2   102.2  5048.2  105.47  5098.5  105.73  5118.5  105.19  5158.5  106.22
  5198.5  105.34  5258.5  107.28  5318.5  106.31  5378.5   108.5  5518.5  108.59
  5558.5  107.74  5628.5  110.39  5748.5  110.48  5858.5   111.9  5963.8  111.68
#Mann= 6 ,-1 , 0
  4157.9     .14       0  4707.9      .1       0  4907.9    .045       0
  4937.9     .04       0  5048.2    .045       0  5098.5      .1       0
Bank Sta=4937.9,5048.2
XS Rating Curve= 0
Exp/Cntr=.3,.1

Type RM Length L Ch R = 1 ,11782.60,134,113.6,98
BEGIN DESCRIPTION:
Cross Section K120-00-00-X06
 Detention ponds on right VRR
END DESCRIPTION:
XS GIS Cut Line= 5
      3101200.99      13951967.8      3100287.57     13951769.64
      3100193.23     13951763.29      3099498.83     13952349.86
      3099071.43      13953308.9
#Sta/Elev= 30
  4007.4   110.8  4197.4   111.1  4287.4   108.2  4477.4   108.8  4931.1  103.02
  4960.2  103.34  4993.5   94.67  4999.4   89.96    5003   90.54  5003.5   92.57
  5007.6   95.26  5017.8   96.34  5039.8  104.18  5066.6   102.6  5526.2   105.9
  5586.6    99.3  5766.6    97.8  5806.6   100.8  5831.2  105.89  5926.6     111
  6025.6   108.6  6206.2  108.87  6295.6    99.7  6515.6   100.5    6557  108.95
  6585.6   111.7  6645.6   110.5  6715.6   112.9  6855.6   110.5  6995.6     112
#Mann= 10 ,-1 , 0
  4007.4     .14       0  4287.4      .1       0  4931.1    .045       0
  4960.2     .04       0  5039.8    .045       0  5066.6      .1       0
  5526.2    .026       0  5831.2      .1       0  6206.2    .026       0
    6557     .99       0
#Block Obstruct= 2 ,-1
    5527    5840  105.91    6206    6560  108.92
Bank Sta=4960.2,5039.8
XS Rating Curve= 0
Exp/Cntr=.3,.1
